--- Case.prj (project) ---

Proj Title=A2C-EA2
Current Plan=p01
Default Exp/Contr=0.3,0.1
SI Units
Geom File=g01
Unsteady File=u01
Plan File=p01
Y Axis Title=Elevation
X Axis Title(PF)=Main Channel Distance
X Axis Title(XS)=Station
BEGIN DESCRIPTION:
A2C-EA2
END DESCRIPTION:
DSS File=dss

--- Case.p01 (plan) ---

Plan Title=Main
Program Version=6.60
Short Identifier=main
Simulation Date=01JAN2000,0000,03JAN2000,0000
Geom File=g01
Flow File=u01
Subcritical Flow
K Sum by GR= 0
Std Step Tol= 0.01
Critical Tol= 0.01
Num of Std Step Trials= 20
Max Error Tol= 0.3
Flow Tol Ratio= 0.001
Split Flow NTrial= 30
Split Flow Tol= 0.02
Split Flow Ratio= 0.02
Log Output Level= 0
Friction Slope Method= 1
Unsteady Friction Slope Method= 2
Unsteady Bridges Friction Slope Method= 1
Parabolic Critical Depth
Global Vel Dist= 0 , 0 , 0
Global Log Level= 0
CheckData=True
Encroach Param=-1 ,0,0, 0
Computation Interval=1SEC
Output Interval=5MIN
Instantaneous Interval=1HOUR
Mapping Interval=5MIN
Computation Time Step Use Courant=        -1
Computation Time Step Use Time Series=    0
Computation Time Step Max Courant=1
Computation Time Step Min Courant=0.45
Computation Time Step Count To Double=4
Computation Time Step Max Doubling=3
Computation Time Step Max Halving=6
Computation Time Step Residence Courant=0
Run HTab=-1
Run UNet=-1
Run Sediment= 0
Run PostProcess= 0
Run WQNet= 0
Run RASMapper= 0
UNET Theta= 1
UNET Theta Warmup= 1
UNET ZTol= 0.02
UNET ZSATol= 0.02
UNET MxIter= 20
UNET Max Iter WO Improvement= 0
UNET MaxInSteps= 0
UNET DtIC= 0
UNET DtMin= 0
UNET MaxCRTS= 20
UNET WFStab= 2
UNET SFStab= 1
UNET WFX= 1
UNET SFX= 1
UNET Gravity=9.81
UNET 1D Methodology=Finite Difference
UNET DSS MLevel= 4
UNET Pardiso=0
UNET DZMax Abort= 100
UNET Use Existing IB Tables=-1
UNET Froude Reduction=False
UNET Froude Limit= 1
UNET Froude Power= 10
UNET D1 Cores= 0
UNET D2 Coriolis=0
UNET D2 Theta= 1
UNET D2 Theta Warmup= 1
UNET D2 Z Tol= 0.01
UNET D2 Volume Tol= 0.01
UNET D2 Max Iterations= 20
UNET D2 Equation= 2
UNET D2 RampUpFraction=0.1
UNET D2 TimeSlices= 1
UNET D2 Turbulence Formulation=None
UNET D2 BCVolumeCheck=0
UNET D2 Cores=0
UNET D2 SolverType=Pardiso (Direct)
UNET D2 Name=Strip
UNET D2 Coriolis=0
UNET D2 Theta= 1
UNET D2 Theta Warmup= 1
UNET D2 Z Tol= 0.01
UNET D2 Volume Tol= 0.01
UNET D2 Max Iterations= 20
UNET D2 Equation= 2
UNET D2 RampUpFraction=0.1
UNET D2 TimeSlices= 1
UNET D2 Turbulence Formulation=None
UNET D2 BCVolumeCheck=0
UNET D2 Cores=0
UNET D2 SolverType=Pardiso (Direct)
UNET D1D2 MaxIter= 0
UNET D1D2 ZTol=0.02
UNET D1D2 QTol=1
DSS File=dss
Write IC File= 0
Write IC File at Fixed DateTime=0
Write IC File at Sim End=0
Echo Input=False
Echo Parameters=False
Echo Output=False
Write Detailed= 0
HDF Write Warmup=0
HDF Write Time Slices=0
HDF Flush=0
HDF Additional Output Variable=Cell Velocity
HDF Additional Output Variable=Face Flow
HDF Compression= 1
HDF Chunk Size= 1
HDF Spatial Parts= 1
HDF Use Max Rows=0
HDF Fixed Rows= 1

--- Case.u01 (unsteady flow) ---

Flow Title=main
Program Version=6.60
Use Restart= 0
Boundary Location=                ,                ,        ,        ,                ,Strip           ,                ,Inflow
Interval=1MIN
Flow Hydrograph= 2882
  0.0000  0.0000  0.0000  0.0000  0.0000  0.0000  4.0000  8.0000 12.0000 16.0000
 20.0000 20.0000 20.0000 20.0000 20.0000 20.0000 20.0000 20.0000 20.0000 20.0000
 20.0000 20.0000 20.0000 20.0000 20.0000 20.0000 20.0000 20.0000 20.0000 20.0000
 20.0000 20.0000 20.0000 20.0000 20.0000 20.0000 20.0000 20.0000 20.0000 20.0000
 20.0000 20.0000 20.0000 20.0000 20.0000 20.0000 20.0000 20.0000 20.0000 20.0000
 20.0000 20.0000 20.0000 20.0000 20.0000 20.0000 20.0000 20.0000 20.0000 20.0000
 20.0000 20.0000 20.0000 20.0000 20.0000 20.0000 20.0000 20.0000 20.0000 20.0000
 20.0000 20.0000 20.0000 20.0000 20.0000 20.0000 20.0000 20.0000 20.0000 20.0000
 20.0000 20.0000 20.0000 20.0000 20.0000 20.0000 20.0000 16.0000 12.0000  8.0000
  4.0000  0.0000  0.0000  0.0000  0.0000  0.0000  0.0000  0.0000  0.0000  0.0000
  0.0000  0.0000  0.0000  0.0000  0.0000  0.0000  0.0000  0.0000  0.0000  0.0000
  0.0000  0.0000  0.0000  0.0000  0.0000  0.0000  0.0000  0.0000  0.0000  0.0000
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Stage Hydrograph TW Check=0
Flow Hydrograph Slope= 0.001
Use DSS=False
Use Fixed Start Time=False
Is Critical Boundary=False
Precipitation Mode=Disable
Wind Mode=No Wind Forces
Met BC=Precipitation|Mode=None
Met BC=Evapotranspiration|Mode=None

--- Case.g01 (geometry) ---

Geom Title=A2C-EA2
Program Version=6.60

Storage Area=Strip           ,500999.99844348046,4000999.9980087793
Storage Area Surface Line= 5
   502000.000679  4001999.996762
   502000.000679  3999999.999255
   499999.996208  3999999.999255
   499999.996208  4001999.996762
   502000.000679  4001999.996762
Storage Area Type= 0
Storage Area Is2D=-1
Storage Area Point Generation Data=,,20,20
Storage Area 2D Points= 10000
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Storage Area Mannings=0.03
2D Cell Volume Filter Tolerance=0.003
2D Cell Minimum Area Fraction=0.01
2D Face Profile Filter Tolerance=0.003
2D Face Area Elevation Profile Filter Tolerance=0.003
2D Face Area Elevation Conveyance Ratio=0.02
2D Face Area Laminar Depth=0.2

BC Line Name=Inflow
BC Line Storage Area=Strip
BC Line Start Position= 500000.0 , 4002000.0
BC Line Middle Position= 500000.0 , 4001950.0
BC Line End Position= 500000.0 , 4001900.0
BC Line Arc= 2
   500000.000000  4002000.000000   500000.000000  4001900.000000
LCMann Table=0

Chan Stop Cuts=-1
